--- TILHANCECK.prj (project) ---

Proj Title=TILHANCECK
Current Plan=p01
Default Exp/Contr=0,0
English Units
Geom File=g01
Flow File=f01
Plan File=p01
BEGIN DESCRIPTION:
END DESCRIPTION:
DSS Export Rating Curves= 0
DSS Export Rating Curve Sorted= 0
DSS Export Volume Flow Curves= 0
DXF OffsetX= 0
DXF OffsetY= 0
DXF ScaleX= 0
DXF ScaleY= 0

--- TILHANCECK.p01 (plan) ---

Plan Title=Floodplain
Program Version=4.00
Geom File=g01
Flow File=f01
K Sum by GR=0
Std Step Tol=0.01
Critical Tol=0.01
Num of Std Step Trials=20
Max Error Tol=0.3
Flow Tol Ratio=0.001
Split Flow NTrial=30
Split Flow Tol=0.02
Split Flow Ratio=0.02
Log Output Level=0
Friction Slope Method=1
Unsteady Friction Slope Method=2
Unsteady Bridges Friction Slope Method=1
Global Log Level=0
CheckData=False
Run HTab=0
Run UNet=0
Run PostProcess=0
UNET Theta=0
UNET Theta Warmup=0
UNET ZTol=0
UNET ZSATol=0
UNET MxIter=0
UNET MaxInSteps=0
UNET DtIC=0
UNET DtMin=0
UNET MaxCRTS=0
UNET WFStab=0
UNET SFStab=0
UNET WFX=0
UNET SFX=0
UNET DSS MLevel=0
UNET DZMax Abort=0
UNET Convert EG Bridges=0
UNET Use Existing IB Tables=0
UNET Froude Limit=0
UNET Froude Power=0
Write IC File=0
Echo Input=False
Echo Output=False
Write Detailed=0

--- TILHANCECK.f01 (steady flow) ---

Flow Title=NFF Regression Equation
Program Version=4.00
Number of Profiles=1
Profile Names=P100yr
River Rch & RM=TILHANCECK,Main      ,50669
421.6794
River Rch & RM=TILHANCECK,Main      ,50035.4
598.6324
River Rch & RM=TILHANCECK,Main      ,49498.9
637.7650
River Rch & RM=TILHANCECK,Main      ,45882.3
697.0285
River Rch & RM=TILHANCECK,Main      ,45582.3
869.2987
River Rch & RM=TILHANCECK,Main      ,44387.1
877.6572
River Rch & RM=TILHANCECK,Main      ,43742.4
1103.202
River Rch & RM=TILHANCECK,Main      ,43427.7
1112.745
River Rch & RM=TILHANCECK,Main      ,39935
1231.282
River Rch & RM=TILHANCECK,Main      ,33339.5
1784.343
River Rch & RM=TILHANCECK,Main      ,33339.5
1333.025
River Rch & RM=TILHANCECK,Main      ,28490.1
1895.675
River Rch & RM=TILHANCECK,Main      ,26523.7
2100.523
River Rch & RM=TILHANCECK,Main      ,26297.3
3171.008
River Rch & RM=TILHANCECK,Main      ,23648.4
3243.297
River Rch & RM=TILHANCECK,Main      ,19954.4
3594.610
River Rch & RM=TILHANCECK,Main      ,407
3968.383
River Rch & RM=TILHANCECK,Main      ,157.1
3969.176
Boundary for River Rch & Prof#=TILHANCECK,Main      ,1
Up Type=0
Dn Type=3
Dn Slope=0.002427

--- TILHANCECK.g01 (geometry) ---

Geom Title=USGS 10m DEM
Program Version=4.10

River Reach=TILHANCECK      ,Main
Reach XY= 30
     2363733.851      376447.816     2364353.999      376702.544
     2365732.115       379954.76     2366358.851      380180.455
     2367640.102      381959.969     2368699.129       384454.76
     2368306.768      385062.399     2369277.254       386352.33
      2370426.56       386111.01      2371505.07      386630.952
      2372622.74      386303.719     2372692.185      387143.996
     2373681.768      388685.663     2373438.713      388918.302
      2373770.31      389810.663     2375251.213      391494.691
     2377141.837      395296.774     2378879.685       396392.26
     2379905.726      396076.288     2379798.087      394961.704
     2380096.699      394671.774     2383633.157      394965.177
     2384226.907      395612.746      2383935.24      397145.732
     2385204.337       397946.08     2386650.518      398246.427
     2387074.129      400390.524     2388577.601      399810.663
     2388850.171      400433.927     2390570.557      400339.945

Type RM Length L Ch R = 1 ,50669   ,205.5,223.6,241.6
XS GIS Cut Line= 3
     2363817.559      376737.257     2363760.267      376645.243
     2363687.014      376016.089
#Sta/Elev= 30
       0  699.85    15.5  697.11    34.8     687    73.6  674.49   124.3   654.9
  137.19652.1655   184.1     650  202.27 646.223     212  645.03   247.8  645.08
   267.7   643.8   283.7  645.64   295.6  645.55  301.32  644.36   307.6  643.41
   315.5  644.25   331.5  646.59   379.3  647.58   403.2  646.97  448.66649.6351
     459  649.12  464.99651.3659   482.9   659.8   498.8  669.46   546.6  690.04
   578.5  706.76   598.4  713.87   622.3  720.84   666.1  729.45   741.8  739.65
#Mann= 7 ,-1 , 0
       0     .12       0  137.19    .016       0  202.27     .12       0
  301.32    .045       0   315.5     .12       0  448.66    .016       0
  464.99     .12       0
#XS Ineff= 2 , 0
          244.42  648.04
Permanent Ineff=
       F       F
Bank Sta=301.32,315.5
XS Rating Curve= 0 ,0
Exp/Cntr=0.3,0.1

Type RM Length L Ch R = 1 ,50445.5 ,41.9,41.9,41.9
XS GIS Cut Line= 4
     2363768.947      376544.549     2363900.892      376466.424
     2363985.961      376357.049     2364121.378      376136.563
#Sta/Elev= 30
       0  648.15   22.69646.8674    47.2  645.69      59   645.5    78.6   644.4
   110.1  643.59   160.5 643.718   173.1  643.21     185  643.29     189  643.06
   196.9  641.76   200.8  641.49   212.7  642.02   220.6  641.68   224.6  641.87
   248.4  643.38  279.36644.3321   311.8  645.68   319.8   645.1  345.43645.2749
  358.39645.5767  387.77646.4565   415.8646.7612   435.2   646.9  468.22648.6677
     487  650.44  527.38657.5497   538.7  659.12  545.62659.4238   550.6  659.72
#Mann= 13 ,-1 , 0
       0     .06       0   22.69    .016       0   160.5     .12       0
   196.9    .045       0   224.6     .06       0  279.36    .016       0
  345.43     .06       0  358.39    .016       0  387.77     .06       0
   415.8    .016       0  468.22     .12       0  527.38     .06       0
  545.62     .12       0
#XS Ineff= 2 , 0
          120.15   645.2  260.33          645.61
Permanent Ineff=
       F       F
Bank Sta=196.9,224.6
XS Rating Curve= 0 ,0
Exp/Cntr=0.3,0.1

Type RM Length L Ch R = 1 ,50403.6 ,54.8,53.3,51.9
XS GIS Cut Line= 4
     2363789.781      376582.743     2363921.725      376504.618
     2364006.795      376395.243     2364142.211      376174.757
#Sta/Elev= 30
       0  648.16    11.8  646.94    43.2  645.22    78.6  644.44    98.3   644.3
  113.02643.7228  135.33  643.33   157.3  643.04   165.2  643.43  171.99644.2935
   177.1   644.9     181  644.98   220.6  645.13   224.6  645.01   228.6  644.26
  231.07  643.09   236.5   641.9   248.5  643.11   256.3  644.25   260.2  644.49
   291.9  644.48  437.77646.2014  462.99646.5986   490.9  647.13  496.13649.1773
   502.9  652.63   506.9   653.9   514.8   655.6  522.87656.1938   550.6  658.02
#Mann= 10 ,-1 , 0
       0     .12       0  113.02    .016       0  135.33     .06       0
  171.99    .016       0  231.07    .045       0   248.5    .016       0
  437.77     .12       0  462.99    .016       0  496.13     .12       0
  522.87     .06       0
#XS Ineff= 2 , 0
          200.26  646.02
Permanent Ineff=
       F       F
Bank Sta=231.07,248.5
XS Rating Curve= 0 ,0
Exp/Cntr=0.3,0.1

Type RM Length L Ch R = 1 ,50350.3 ,78.3,78.3,78.3
XS GIS Cut Line= 3
     2363948.418         376660.      2363985.31      376514.601
     2364168.687      376248.759
#Sta/Elev= 30
       0  687.06   13.99684.4955    19.7  683.52    31.6  679.18    43.4  676.27
    67.1  671.45    90.8  667.36    98.7  665.39   110.5  660.76   126.3  653.43
     150  644.62     166  642.26  176.24642.5928   181.9  642.29   189.9  639.85
   193.9  638.86   205.8   638.6   219.9  639.34  240.08641.5223   249.7  642.37
   273.6   641.9   317.5  643.34   369.3  643.51   399.1 644.279  420.14 645.736
   433.1  645.27     453  645.73     457  647.01  466.12653.1372     473  655.04
#Mann= 9 ,-1 , 0
       0     .12       0   13.99     .06       0  176.24     .12       0
   189.9    .045       0   219.9     .12       0  240.08     .06       0
   399.1     .12       0  420.14    .016       0  466.12     .12       0
Bank Sta=189.9,219.9
XS Rating Curve= 0 ,0
Exp/Cntr=0.3,0.1

Type RM Length L Ch R = 1 ,50272   ,71.9,75.3,78.6
XS GIS Cut Line= 3
     2364011.352      376706.658     2364048.244      376561.259
     2364231.621      376295.417
#Sta/Elev= 30
       0  687.73    67.1  677.34      79  673.71    86.8  670.43    98.7  668.03
   110.5  664.53   130.3  655.46   138.2  653.39     150  652.84     162  647.67
   185.9  640.29   193.9  638.72   205.8  637.96   221.5  638.61   225.8  640.14
   233.7  644.68   237.7  646.04   241.7  645.77   249.7  641.97   253.7   640.9
   261.6  640.04   316.2640.3928   361.3  640.39  417.35641.9763   441.1  642.34
  445.93643.9406     453  648.45     457  650.09     465  652.08     473  653.19
#Mann= 6 ,-1 , 0
       0     .12       0   193.9    .045       0   221.5     .12       0
   316.2     .06       0  417.35    .016       0  445.93     .12       0
#XS Ineff= 2 , 0
                          240.05           647.6
Permanent Ineff=
       F       F
Bank Sta=193.9,221.5
XS Rating Curve= 0 ,0
Exp/Cntr=0.3,0.1

Type RM Length L Ch R = 1 ,50196.7 ,155.6,161.3,165.8
XS GIS Cut Line= 3
     2364033.647      376718.189     2364075.313      376625.741
     2364416.083       376257.44
#Sta/Elev= 30
       0  689.36    15.6  686.26    42.9  679.56      78   669.9    97.5  663.79
   125.3  650.89   145.2  643.17   172.3  638.46     181  637.96   187.3  638.82
     197  639.82   216.9  639.27   232.8  640.28   244.8  640.18   256.7  638.58
  324.11637.9758  358.69639.5522   380.2  639.14   400.1  640.06   408.2639.6646
   431.9  641.78   435.9  642.73   439.9  644.21   451.8  649.66   479.7  658.41
   491.7  662.72   543.4  683.76   551.4  686.47   575.3  693.38   603.2   703.3
#Mann= 6 ,-1 , 0
       0     .12       0   172.3    .045       0   187.3     .12       0
  324.11     .06       0  358.69    .016       0   408.2     .12       0
#XS Ineff= 2 , 0
                          332.48          641.63
Permanent Ineff=
       F       F
Bank Sta=172.3,187.3
XS Rating Curve= 0 ,0
Exp/Cntr=0.3,0.1

Type RM Length L Ch R = 1 ,50035.4 ,106.4,108.1,106.4
XS GIS Cut Line= 2
     2364083.126      376787.199     2364443.803      376500.741
#Sta/Elev= 30
       0  681.56    15.9  676.25    47.6  662.14    63.5  656.18    71.5  653.66
    83.4  648.31   107.2  645.51   146.9   638.6   170.7  638.01   182.6  637.19
   202.5  638.03   210.3  636.78   214.4  635.74   218.4  635.36   225.3  636.13
   232.7 637.422     266  637.56   293.8   636.6   301.8  635.88   313.7  636.45
   321.6  635.88   333.5     637   353.4  637.98   365.3  639.23   389.1  639.68
   393.1  641.41  399.57645.7073   416.9  653.05   428.8  657.38   460.6  671.57
#Mann= 5 ,-1 , 0
       0     .12       0   210.3    .045       0   225.3     .12       0
   232.7    .016       0  399.57     .12       0
#XS Ineff= 2 , 0
                          288.83          640.56
Permanent Ineff=
       F       F
Bank Sta=210.3,225.3
XS Rating Curve= 0 ,0
Exp/Cntr=0.3,0.1

Type RM Length L Ch R = 1 ,49927.3 ,169.2,176.4,181.3
XS GIS Cut Line= 2
     2364130.001      376851.002     2364490.678      376585.377
#Sta/Elev= 30
       0  670.48      20  661.93   32.42657.8129      44  654.03      52  650.76
   68.45649.3491      80  647.21   94.51643.5615     132  637.09     160  635.97
     228  634.66     252  635.28   259.4  634.16     268  633.18   274.4  633.54
  278.56  634.19     292  635.46     316  635.08     340  635.77     348  636.67
     356  639.65     360  640.38  370.55640.9515   403.9  640.94   407.9  641.85
   411.9  644.27   415.9  647.53   431.9  662.52   435.9  665.54   447.9  670.63
#Mann= 8 ,-1 , 0
       0    .016       0   32.42     .12       0   68.45     .06       0
   94.51     .12       0   259.4    .045       0   274.4     .12       0
  370.55    .016       0   403.9     .12       0
#XS Ineff= 2 , 0
                          326.06          638.09
Permanent Ineff=
       F       F
Bank Sta=259.4,278.56
XS Rating Curve= 0 ,0
Exp/Cntr=0.3,0.1

Type RM Length L Ch R = 1 ,49751   ,358.3,252,254.3
XS GIS Cut Line= 3
     2364079.219      376964.283     2364549.738      376784.542
     2364688.594      376815.845
#Sta/Elev= 30
       0  712.06       4  710.93      16  704.42      36  696.82      68  682.66
   143.9  646.99   151.9   642.1   155.9  640.46   187.9  635.47   215.9   633.3
   323.8  632.91   327.8  632.82  333.42  631.72   339.8   630.6   347.8  630.83
   351.8  632.17   355.8  633.45   359.8   633.7   427.7  633.53   447.7  634.43
   451.7  635.36   463.7  640.34   475.7  642.99   487.7  644.75   495.7  648.05
   539.3  662.12     559  669.37   582.8  675.52   618.3  686.01     646  691.56
#Mann= 3 ,-1 , 0
       0     .12       0  333.42    .045       0   351.8     .12       0
#XS Ineff= 2 , 0
                          394.48          639.26
Permanent Ineff=
       F       F
Bank Sta=333.42,351.8
XS Rating Curve= 0 ,0
Exp/Cntr=0.3,0.1

Type RM Length L Ch R = 1 ,49498.9 ,197.9,305.2,302.5
XS GIS Cut Line= 3
     2363977.873       377162.55      2364473.41      377062.376
     2364853.285      376963.438
#Sta/Elev= 30
       0  720.79    43.8  720.54   88.21716.0542  125.43714.7297   175.2  710.94
     203  703.71   234.9  692.22   290.6  668.03   346.3  639.87   366.2  632.75
   386.1  627.82   398.1  630.25     418  628.06   433.9  628.81   441.9  627.95
   457.8  629.91   501.6  629.09   509.5  627.99   517.5   629.2   553.1  633.25
   576.9  633.67   604.7   636.3   632.4  645.39     684  667.25   719.7  678.26
   731.6  680.48   771.2  691.83     803  699.57   878.3  716.09   898.1  718.43
#Mann= 5 ,-1 , 0
       0    .016       0   88.21     .06       0  125.43     .12       0
   501.6    .045       0   517.5     .12       0
Bank Sta=501.6,517.5
XS Rating Curve= 0 ,0
Exp/Cntr=0.3,0.1

Type RM Length L Ch R = 1 ,49193.7 ,318.1,310.4,303.3
XS GIS Cut Line= 2
      2364248.49      377296.314     2364830.522      377114.022
#Sta/Elev= 30
       0   683.3      16  680.65    35.9  675.89    47.8  672.25    79.7  660.85
    91.7  655.64   131.6  634.06   143.5  628.53   147.5  627.46   151.5  627.08
   167.4  626.86   176.9  625.53   191.3  624.82   195.3  625.37   203.3     628
   207.3  628.63   227.2  627.58   259.1  628.54     279  628.54     299  630.24
   334.8  629.98   370.7  631.17   386.7  633.02   402.6  636.24   410.6  638.74
   474.4  666.13   498.3   675.7   530.2  684.17     574  697.37   609.9  706.08
#Mann= 3 ,-1 , 0
       0     .12       0   176.9    .045       0   195.3     .12       0
Bank Sta=176.9,195.3
XS Rating Curve= 0 ,0
Exp/Cntr=0.3,0.1

Type RM Length L Ch R = 1 ,48883.4 ,223,231.3,234.9
XS GIS Cut Line= 2
     2364347.449      377660.897     2364907.105      377246.133
#Sta/Elev= 30
       0  706.92    27.9  701.84    47.8  696.61    75.6  687.26   107.5  674.74
   127.4  666.01   151.3  653.74   183.1  634.65     199  626.25     203  625.01
     207  624.72   226.9  625.19   237.4  623.54   250.8  622.95  255.49  623.69
   262.7  625.59   270.7   625.8   290.6   624.4   334.4  624.87   346.3  626.32
   354.3  626.02   429.9   629.6   445.8  631.52   469.7  639.16   533.4  668.29
   557.3  676.66   589.1  685.67     613  690.83   684.6  708.77   696.6  710.98
#Mann= 3 ,-1 , 0
       0     .12       0   237.4    .045       0  255.49     .12       0
Bank Sta=237.4,255.49
XS Rating Curve= 0 ,0
Exp/Cntr=0.3,0.1

Type RM Length L Ch R = 1 ,48652   ,367,372,377.7
XS GIS Cut Line= 2
     2364452.917      377783.293     2364990.678      377483.814
#Sta/Elev= 30
       0  694.62      24     687      44  678.78      52  676.69      68  669.79
   135.9  638.96   155.9  628.68   163.9   623.3   167.9  622.09   183.9  623.49
   203.8  622.94   219.8  623.83   243.8  623.15   267.8  623.83   279.8  622.12
   303.8  622.46   315.8   621.8   323.8  620.86   331.8  621.68   343.7  622.71
   359.7  622.07   375.7  625.39   383.7  625.29   391.7  626.46   407.7  632.03
   447.7  652.08   495.6  669.56   543.6  681.58   575.6  686.81   615.5  691.54
#Mann= 3 ,-1 , 0
       0     .12       0   315.8    .045       0   331.8     .12       0
Bank Sta=315.8,331.8
XS Rating Curve= 0 ,0
Exp/Cntr=0.3,0.1

Type RM Length L Ch R = 1 ,48280   ,332.7,329.7,324.9
XS GIS Cut Line= 2
     2364562.292      378026.783     2365170.365      377823.658
#Sta/Elev= 30
       0  654.45    27.9  653.09    39.8  650.04   54.62648.0419   70.18644.2364
   103.5  638.44   111.5  634.13   131.4  628.21   163.3  624.12   183.2  620.41
   203.1  619.96     215  621.15   234.9  617.69   246.9   618.6   282.7  618.97
   301.7  617.02   314.6  616.52   322.5  616.94   330.5  617.55   346.4  620.46
   362.4  621.82   370.3  621.24   378.3  622.09   398.2  629.07   457.9  657.04
   513.7   677.3   537.6  684.56   561.5  690.76   581.4  695.01   641.1  705.31
#Mann= 5 ,-1 , 0
       0     .12       0   54.62     .06       0   70.18     .12       0
   301.7    .045       0   322.5     .12       0
#XS Ineff= 2 , 0
          215.66  622.81
Permanent Ineff=
       F       F
Bank Sta=301.7,322.5
XS Rating Curve= 0 ,0
Exp/Cntr=0.3,0.1

Type RM Length L Ch R = 1 ,47950.3 ,203.3,203.4,203.8
XS GIS Cut Line= 3
     2364611.772      378249.439     2365036.251      378073.658
     2365126.094      377943.449
#Sta/Elev= 30
       0   689.7    47.9  674.05    67.9  666.71    95.9  655.46   151.8  631.56
   159.8  627.49   167.8  625.47   175.8  622.37   191.8  618.08   235.7  616.14
   242.7  613.77   247.7  612.68   257.7  613.67   271.7  616.04   291.6  615.37
   327.6  616.02   343.6  614.56   359.6  613.95   363.6  614.25   387.5  619.54
   403.5  620.25   431.5   623.5   443.5  626.07   455.4  629.95   491.1  645.66
   514.8  654.11   554.4   666.1     582  672.91   597.9  678.42   617.6  682.56
#Mann= 3 ,-1 , 0
       0     .12       0   242.7    .045       0   257.7     .12       0
Bank Sta=242.7,257.7
XS Rating Curve= 0 ,0
Exp/Cntr=0.3,0.1

Type RM Length L Ch R = 1 ,47746.9 ,361,361.6,353.7
XS GIS Cut Line= 3
     2364709.428      378414.804     2365126.094      378250.741
     2365291.459      378240.324
#Sta/Elev= 30
       0  674.87      48  653.33     100   627.8     112  622.77     124  618.95
   131.9  617.61   151.9  616.06   199.9  614.82   211.9  614.34   223.9  613.19
   239.9   613.7   251.9   612.8     265  612.76   275.9  611.44   279.9  611.49
  286.57  612.74   295.9  613.92   311.9  613.08   351.8  614.16   367.8  614.14
   383.8  615.02   387.8  615.83   399.8  619.57   435.8  634.99   487.2  654.71
   518.8   665.6   534.6  670.05     574  678.98   593.8  683.08   613.5  686.37
#Mann= 3 ,-1 , 0
       0     .12       0     265    .045       0  286.57     .12       0
#XS Ineff= 2 , 0
          204.88  616.73
Permanent Ineff=
       F       F
Bank Sta=265,286.57
XS Rating Curve= 0 ,0
Exp/Cntr=0.3,0.1

Type RM Length L Ch R = 1 ,47385.2 ,304.1,301.7,299
XS GIS Cut Line= 3
     2364697.041      378732.094      2365077.92      378577.555
     2365474.156      378430.665
#Sta/Elev= 30
       0  694.16    31.9  693.82    63.8  691.26    87.8  687.23    99.8   683.8
   115.7  677.85   139.7  667.37   175.6  648.93   219.5  624.55   235.4  618.31
   243.4   616.1   255.4  614.51   315.3  613.63   331.2  608.98   383.1  610.88
   403.5  609.69     415   608.5     427  609.74     435   611.5   442.9  612.02
   478.8  611.95   494.8  610.64   514.7  611.97   522.7  614.76   590.4  643.86
   622.3  655.67   654.2  664.97   678.1  670.85   753.9  686.37   833.6  695.18
#Mann= 3 ,-1 , 0
       0     .12       0   403.5    .045       0     427     .12       0
#XS Ineff= 2 , 0
                          450.58           613.9
Permanent Ineff=
       F       F
Bank Sta=403.5,427
XS Rating Curve= 0 ,0
Exp/Cntr=0.3,0.1

Type RM Length L Ch R = 1 ,47083.6 ,263.1,265.9,263.7
XS GIS Cut Line= 3
      2364778.78       379026.98     2365134.263      378836.971
     2365538.619      378650.994
#Sta/Elev= 30
       0  671.96      24  670.57    63.8   666.3   139.7  654.18   167.6  648.57
   207.5  636.68   251.4  626.95   311.3  617.09   339.2  614.14   371.2  612.16
   379.1  610.81  388.72  606.49   391.1  605.29   399.1     605     415  605.26
  420.69  606.38   442.8  608.04   470.6  607.69   506.4  608.26   522.3   610.1
     574  613.55   593.8  615.83   609.7  618.22   641.5  625.42   673.3  631.47
   701.1  638.29     721  642.37   740.9  645.34   800.5  651.22   848.2  658.32
#Mann= 3 ,-1 , 0
       0     .12       0  388.72    .045       0  420.69     .12       0
Bank Sta=388.72,420.69
XS Rating Curve= 0 ,0
Exp/Cntr=0.3,0.1

Type RM Length L Ch R = 1 ,46817.7 ,137.6,139.4,140.4
XS GIS Cut Line= 2
     2364964.636      379133.554     2365597.449      378895.272
#Sta/Elev= 30
       0  682.53    23.9   678.7    55.7  671.46    79.6  665.06   111.4  653.44
     171   627.2   202.9  614.42   222.7  609.11   230.7  607.91   250.6   608.6
   262.5   606.9   274.4  606.16   306.3  605.14   330.1  605.76     350  604.46
     358   603.2   365.9  604.26   373.9   605.4   385.8  604.17   401.7  606.92
   453.4  608.72   469.4   609.9   477.3  611.24   485.3  613.84   497.2     619
   517.1  628.82   568.8  652.36   628.5  673.54   664.2  683.11   676.2  685.43
#Mann= 3 ,-1 , 0
       0     .12       0     350    .045       0   365.9     .12       0
Bank Sta=350,365.9
XS Rating Curve= 0 ,0
Exp/Cntr=0.3,0.1

Type RM Length L Ch R = 1 ,46678.3 ,45.7,45.7,45.7
XS GIS Cut Line= 2
     2364994.844      379223.137     2365627.657      378984.856
#Sta/Elev= 30
       0  675.12    59.7  663.48   131.3  644.67     187   628.4   210.8   620.5
   214.8  618.52   222.7  611.77   226.7  609.87   234.7  608.88  251.01608.8567
  259.54608.4778   262.5  608.13   270.5  604.68   291.4  603.11   298.3  602.03
   306.4  603.24   318.2  605.06   342.1  605.98   369.9  604.28   389.8   605.6
   469.4  607.35   505.2  609.38   509.1  610.18   513.1  612.08     525  620.73
     537   626.8   596.6   654.3   620.5  662.33   656.3  671.85   676.2  676.36
#Mann= 5 ,-1 , 0
       0     .12       0  251.01    .016       0  259.54     .12       0
   291.4    .045       0   306.4     .12       0
Bank Sta=291.4,306.4
XS Rating Curve= 0 ,0
Exp/Cntr=0.3,0.1

Type RM Length L Ch R = 1 ,46632.6 ,169.3,169.2,169.3
XS GIS Cut Line= 2
     2365015.157      379264.283     2365647.969      379026.002
#Sta/Elev= 30
       0  664.12   103.4  638.59   123.3  634.14   143.2  630.41     183  624.92
   202.9  621.49   206.8  620.23   218.8  611.38   222.7  609.99  232.81609.6944
   246.6  609.77  258.56609.0732   274.4  606.91   288.3  601.41   298.3  600.24
   306.3  600.67   310.2  601.86   314.2  603.46   318.2  603.96     346  603.06
   405.7  603.84   449.5  606.86   481.3  606.99   493.2  608.17   513.1  613.76
   560.8   635.3   592.7  648.22   604.6  652.24   628.5  658.53   676.2  667.96
#Mann= 5 ,-1 , 0
       0     .12       0  232.81    .016       0  258.56     .12       0
   288.3    .045       0   310.2     .12       0
Bank Sta=288.3,310.2
XS Rating Curve= 0 ,0
Exp/Cntr=0.3,0.1

Type RM Length L Ch R = 1 ,46463.4 ,182,180.5,178.9
XS GIS Cut Line= 2
     2365119.931      379405.081     2365731.436      379175.327
#Sta/Elev= 30
       0  671.41    35.8  668.62    59.8  665.53    79.7  661.43    95.6  657.12
   107.6  652.96   143.4   636.8   179.2  616.04  184.72612.3576   191.2  607.67
   195.2  605.83   215.1  605.07  223.17602.7343     231  600.33     243  599.94
   249.4  600.38   258.9  601.58   274.8  600.77   342.6  599.94   382.4  603.65
   414.2  604.47   426.2  604.31   446.1  605.69   454.1  606.76     486  615.22
   497.9  619.11   577.6  647.99   613.4  661.82   629.3  666.41   653.2  672.41
#Mann= 5 ,-1 , 0
       0     .12       0  184.72    .016       0  223.17     .12       0
     231    .045       0   249.4     .12       0
Bank Sta=231,249.4
XS Rating Curve= 0 ,0
Exp/Cntr=0.3,0.1

Type RM Length L Ch R = 1 ,46282.9 ,207.7,203.1,198.5
XS GIS Cut Line= 3
     2365208.907      379501.653     2365340.514      379518.609
     2365856.891      379280.586
#Sta/Elev= 30
       0  673.97    23.4  668.25    54.6  656.29    74.2  647.81   132.7  620.04
   148.6  611.76  166.01604.0029   172.5  602.54   188.4   602.4  213.21600.3667
   227.2  598.93   232.1   598.6   242.2  599.15     252  600.39   283.8  599.34
   351.4  599.35   355.4  599.73   367.3  603.13     415   602.6   450.8  604.22
   466.7  605.74   474.6  607.64   490.6  613.17   534.3  632.56   566.1  645.46
     578  649.64   625.7  664.19   657.6  675.13   673.5  679.77   701.3  686.42
#Mann= 5 ,-1 , 0
       0     .12       0  166.01    .016       0  213.21     .12       0
   227.2    .045       0   242.2     .12       0
Bank Sta=227.2,242.2
XS Rating Curve= 0 ,0
Exp/Cntr=0.3,0.1

Type RM Length L Ch R = 1 ,46079.7 ,67.3,68.8,70.3
XS GIS Cut Line= 3
     2365230.608       379623.18     2365500.791      379675.264
     2365792.674       379460.42
#Sta/Elev= 30
       0  658.41    63.8  641.86   115.6  624.09   135.6  617.86   155.5  614.61
   163.5  614.49   177.6615.6185   195.4  614.49   215.3  611.42  237.91606.7733
   263.2  602.12     299  599.22     303  598.33     307  596.46     311  595.15
     315  594.87     323  596.22   342.9  597.76  357.05597.9031   478.3  598.87
   490.2  599.78  506.76602.8215     538  603.66   559.8 607.479   577.8     609
   597.8  612.93   601.7  615.21   605.7  619.14   609.7  622.12   637.6  635.81
#Mann= 8 ,-1 , 0
       0     .12       0   177.6     .06       0  237.91    .016       0
     307    .045       0     323    .016       0  357.05     .12       0
  506.76     .08       0   559.8     .12       0
Bank Sta=307,323
XS Rating Curve= 0 ,0
Exp/Cntr=0.3,0.1

Type RM Length L Ch R = 1 ,46011   ,129,128.7,128.4
XS GIS Cut Line= 3
     2365303.308      379802.217     2365523.577      379739.283
     2365854.523      379527.694
#Sta/Elev= 30
       0  664.88    15.8  660.32    63.2  649.21    98.7  639.17   146.1  628.08
   177.7  616.45   209.3  603.31   221.2  599.12  225.76598.7864     241  599.39
   256.9   598.9   264.8  598.05   272.7  595.74   280.7  594.85   291.3  595.82
   312.4  599.81   320.3  600.38   328.3  600.14   336.2  597.83  342.42597.1278
  396.46  597.11   419.5   597.2  452.73601.4744  486.99601.5905   506.8  601.31
   526.7  603.52   538.6  606.21   550.5  609.83   558.4  614.15   621.9  640.68
#Mann= 8 ,-1 , 0
       0     .12       0  225.76    .016       0   272.7    .045       0
   291.3     .12       0  342.42     .04       0  396.46     .12       0
  452.73    .016       0  486.99     .12       0
#XS Ineff= 2 , 0
                          322.59          602.04
Permanent Ineff=
       F       F
Bank Sta=272.7,291.3
XS Rating Curve= 0 ,0
Exp/Cntr=0.3,0.1

Type RM Length L Ch R = 1 ,45882.3 ,309.8,300,292.3
XS GIS Cut Line= 3
      2365300.41       380041.03     2365642.508      379815.951
     2365984.121       379590.14
#Sta/Elev= 30
       0  606.11   29.86606.5091    90.2604.4023     167  602.17   214.7  602.07
  254.32600.9005  308.52 601.473     322  600.55   337.9   598.1   357.8  597.59
   373.7     594   393.6  594.75   397.6  593.92   401.6  592.64   405.5   592.5
   413.5  593.98   429.4  598.49   444.6600.1565  446.03600.1235   461.2  597.12
  609.34  597.11  621.03597.4336     652  603.44     664  603.62  678.13602.5115
   683.8  602.96   687.8  604.13   723.6  617.88   771.3  633.27     819  646.39
#Mann= 12 ,-1 , 0
       0     .12       0   29.86    .016       0    90.2     .12       0
  254.32    .016       0  308.52     .12       0   397.6    .045       0
   413.5     .12       0   444.6     .06       0  446.03     .04       0
  609.34     .12       0  621.03    .016       0  678.13     .12       0
#XS Ineff= 2 , 0
                          446.73          601.71
Permanent Ineff=
       F       F
Bank Sta=397.6,413.5
XS Rating Curve= 0 ,0
Exp/Cntr=0.3,0.1

Type RM Length L Ch R = 1 ,45582.3 ,259.1,254,247.3
XS GIS Cut Line= 3
     2365613.675      380396.961     2365826.199      380049.196
      2366080.39      379714.248
#Sta/Elev= 30
       0   656.1      44  661.04   57.57660.8468    75.9  663.96  111.71665.8905
   151.8  667.21  176.97666.4932  223.05663.2425   247.7  660.23   267.7   655.3
   287.7  651.57   303.7  644.47   327.6  631.79   367.6  607.42  398.02  591.63
   399.6  590.33   407.6  589.57   419.5  591.48   423.4  591.52  453.07598.5912
   463.1  600.15  469.27600.1121   482.9  597.13  741.31597.1902   744.7  597.59
   760.6  603.23   768.5  604.89  787.54604.9714   816.1  606.53     828  611.22
#Mann= 11 ,-1 , 0
       0     .12       0   57.57    .016       0  111.71     .12       0
  176.97    .016       0  223.05     .12       0  398.02    .045       0
   419.5     .12       0  453.07     .06       0  469.27     .04       0
  741.31     .06       0  787.54     .12       0
Bank Sta=398.02,419.5
XS Rating Curve= 0 ,0
Exp/Cntr=0.3,0.1

Type RM Length L Ch R = 1 ,45328.2 ,309.3,320,330
XS GIS Cut Line= 3
     2365969.541      380399.005     2366068.282      380113.632
     2366306.997      379860.811
#Sta/Elev= 30
       0  668.23    43.7  658.25   64.42652.1743   98.48640.9623     143  622.68
   190.7  600.92   202.6  597.27   222.5  592.52   242.4  589.25   254.3  588.18
   264.2  589.33   270.2  589.86   282.1   592.1  300.83597.2497     318  599.68
  335.26599.5466  341.72598.8621   353.9  597.58   365.9  597.13  508.61  597.11
   517.8  597.14   521.8  597.67   529.8  600.98   541.8  602.74   545.8  605.41
   553.8  611.87   585.7  629.28   609.7  641.52   629.7  650.53   649.7  657.23
#Mann= 9 ,-1 , 0
       0     .12       0   64.42    .016       0   98.48     .12       0
   242.4    .045       0   264.2     .12       0  300.83     .04       0
  335.26     .06       0  341.72     .04       0  508.61     .12       0
Bank Sta=242.4,264.2
XS Rating Curve= 0 ,0
Exp/Cntr=0.3,0.1

Type RM Length L Ch R = 1 ,45008.2 ,238.8,238.1,230.5
XS GIS Cut Line= 2
     2366054.176      380467.364     2366586.945      379950.871
#Sta/Elev= 30
       0   659.4   107.7  632.41   151.6  624.41   171.5  621.69   183.5  619.04
   191.5  616.96   235.4  600.47   263.3  594.74   327.1  586.93   339.1  587.97
     363   586.5     371  587.53     391  588.12   398.9  588.03   406.9  586.47
   410.9  586.01   424.8  586.35   434.8  587.44   450.8  587.75   458.8  589.27
   462.8  591.34   474.7  600.78   486.7  608.68   514.6  623.34   538.6  637.76
   578.5  655.46   606.4  665.28   630.3  672.66   702.1  687.25     742  694.32
#Mann= 3 ,-1 , 0
       0     .12       0   406.9    .045       0   424.8     .12       0
Bank Sta=406.9,424.8
XS Rating Curve= 0 ,0
Exp/Cntr=0.3,0.1

Type RM Length L Ch R = 1 ,44770.1 ,379.3,383,387.1
XS GIS Cut Line= 3
      2366269.02      380509.682     2366471.928       380320.88
     2366639.028      380159.205
#Sta/Elev= 30
       0  633.29    15.8  632.96    51.5   628.9    67.3  626.35    91.1  621.04
   118.8   612.6   150.5  598.37   158.4  594.19   178.2  587.65   186.1   586.8
     198  587.03   213.8   586.4   241.5  584.29   257.4  585.16   265.3  584.08
   269.2  584.06  278.91  585.34     285  586.36   296.9   584.3   300.8   584.2
   312.6  585.12   316.6  586.26   340.2  597.74   359.9  609.39   375.7  617.67
   411.2  634.08     423  639.07   438.7  644.72   450.6   648.1   509.7  661.66
#Mann= 3 ,-1 , 0
       0     .12       0   257.4    .045       0  278.91     .12       0
Bank Sta=257.4,278.91
XS Rating Curve= 0 ,0
Exp/Cntr=0.3,0.1

Type RM Length L Ch R = 1 ,44387.1 ,210.7,211.1,211.3
XS GIS Cut Line= 3
     2366430.695      380606.253     2366626.008      380651.826
     2366982.995      380410.941
#Sta/Elev= 30
       0  624.96    43.3  622.39    62.9  620.43   106.2   613.8   121.9  610.45
     177  601.18   192.7  597.56   204.6   593.1   212.5  591.15   232.5  582.69
  246.76  580.37   252.4  579.72   265.3  580.32   272.3  581.64   296.3  582.49
   312.2  580.67   324.2  582.59   340.1   581.7   352.1  581.95     364  584.23
   411.9  588.34   435.8  595.29   455.8  602.34   471.7  605.68   499.6  616.44
   515.6  621.51   539.5  630.97   547.5  633.51   583.4  643.43   631.2  654.57
#Mann= 3 ,-1 , 0
       0     .12       0  246.76    .045       0   265.3     .12       0
Bank Sta=246.76,265.3
XS Rating Curve= 0 ,0
Exp/Cntr=0.3,0.1

Type RM Length L Ch R = 1 ,44176   ,433.8,433.5,430.2
XS GIS Cut Line= 3
     2366627.093       381099.96     2366692.197      380859.074
     2367136.778      380564.294
#Sta/Elev= 30
       0  652.53    87.1  643.78   130.7  635.34   154.5  629.24   190.1  616.68
     206  611.88   249.5  594.84   273.4  586.46   297.3  583.51   317.2  581.98
   333.1   580.9     349  580.77   364.6   577.6   376.9  577.05   380.9  577.48
   396.8  579.44   404.8  581.11   408.8  582.79   436.6  599.53   452.6  605.66
   480.4  612.98   508.3  621.43   552.1  633.52   591.9  641.34   615.8  644.63
   631.7  647.87   659.6   654.6   691.4  663.83   751.1  671.47     783  676.61
#Mann= 3 ,-1 , 0
       0     .12       0   364.6    .045       0   380.9     .12       0
Bank Sta=364.6,380.9
XS Rating Curve= 0 ,0
Exp/Cntr=0.3,0.1

Type RM Length L Ch R = 1 ,43742.4 ,308.5,314.7,320.6
XS GIS Cut Line= 2
      2366819.15      381273.571     2367282.475      380834.118
#Sta/Elev= 30
       0  646.11      12  646.18    31.9  648.21    43.9  645.19    71.8  642.02
    95.8  636.51   127.7  622.88   187.6  590.42   199.6  584.83   215.5  578.78
   231.5  576.43   238.7  574.02   243.5  573.36   253.7  573.91   263.4  576.55
   279.4  575.89   291.4  576.98   335.3  577.47   367.2  577.16   383.2  575.75
   387.1  576.23   399.1  583.14   403.1  584.67     431  592.85     471  603.34
   518.8  614.89   530.8  617.07   554.8  623.44   598.7  637.66   638.6  652.55
#Mann= 3 ,-1 , 0
       0     .12       0   238.7    .045       0   253.7     .12       0
Bank Sta=238.7,253.7
XS Rating Curve= 0 ,0
Exp/Cntr=0.3,0.1

Type RM Length L Ch R = 1 ,43427.7 ,241.6,244,245.7
XS GIS Cut Line= 3
     2366923.317      381303.953     2367122.969      381372.312
     2367511.424      381165.064
#Sta/Elev= 30
       0  635.09      12  633.41    75.6  620.14    99.5   617.2   159.3  612.47
   175.2  609.77   195.1  604.65     211  599.13   266.6   574.8   274.5  573.54
   290.4   574.2   302.3  571.47   310.2  570.49   322.1   571.1     330   573.2
     334  573.41   361.8  572.47   385.6  573.34   393.5  574.25   409.4  572.74
   425.2  575.78   437.1  576.52     457  579.86   468.8   583.9   488.7   593.1
   532.3  615.68   552.2   626.9     568  634.64   607.7   649.4   651.3   669.3
#Mann= 3 ,-1 , 0
       0     .12       0   302.3    .045       0   322.1     .12       0
Bank Sta=302.3,322.1
XS Rating Curve= 0 ,0
Exp/Cntr=0.3,0.1

Type RM Length L Ch R = 1 ,43183.7 ,296.2,295.9,295.3
XS GIS Cut Line= 3
     2366977.631      381671.099     2367361.153      381510.934
     2367741.803      381362.907
#Sta/Elev= 30
       0  641.68      28   641.9   86.51637.5486   115.9  635.05   139.9  631.72
   167.8  625.54   219.8  608.59   251.8  595.17   287.7  577.48   307.7  571.25
   315.7  570.81   331.7  572.04   391.6  572.17   395.6  571.88   407.2  568.91
   419.6  568.54  424.55  569.02   431.5  571.92   435.4  572.72   459.2  574.71
     491  576.19   502.9  579.35   522.7  587.98   554.4  605.08   613.9  639.07
   641.6  653.89   689.2  676.15   732.8  690.86   788.4  707.26     824  713.73
#Mann= 4 ,-1 , 0
       0     .06       0   86.51     .12       0   407.2    .045       0
  424.55     .12       0
Bank Sta=407.2,424.55
XS Rating Curve= 0 ,0
Exp/Cntr=0.3,0.1

Type RM Length L Ch R = 1 ,42887.7 ,328.5,326.4,324
XS GIS Cut Line= 3
      2367131.65      381861.679     2367318.282      381849.743
     2367798.968      381644.665
#Sta/Elev= 30
       0  641.19    31.8  636.39    71.6  626.51    87.5  620.62   143.2  602.68
   218.9   583.7   242.9  576.42   286.8  568.66   322.6  568.79  344.41  566.52
   350.6  566.14   361.2  566.75   370.5  569.68   374.5  570.18   410.4  572.49
   422.4  577.46   454.3  593.99   462.3  597.16  475.86603.9926   506.2  620.19
   530.1     632     554   645.1   593.9  658.19   625.8  671.44   637.8  677.26
   645.8  677.22  677.94 689.205   697.6  696.03   705.6  696.11   709.6  696.95
#Mann= 5 ,-1 , 0
       0     .12       0  344.41    .045       0   361.2     .12       0
  475.86     .06       0  677.94     .12       0
Bank Sta=344.41,361.2
XS Rating Curve= 0 ,0
Exp/Cntr=0.3,0.1

Type RM Length L Ch R = 1 ,42561.4 ,274.3,277.1,280
XS GIS Cut Line= 3
     2367293.325      382059.161     2367404.002      382078.692
     2367795.712      381862.764
#Sta/Elev= 30
       0   607.8    23.2  600.75    34.9  597.64    89.1  580.39    96.9  578.44
   112.4  576.17   152.3  573.45   212.2  570.32   232.2  568.74   240.2  568.76
   248.2  567.97   304.1  567.25     332  568.24     344  568.18     360   565.8
   368.1  563.52     376  562.37     380  562.63   383.1  564.41     384  564.93
     388  570.27   391.9  576.61   395.9  581.51   403.9  589.55   411.9  596.87
   427.9  608.79   475.8  634.46   487.8  641.26   539.7  664.35   559.7   672.1
#Mann= 3 ,-1 , 0
       0     .12       0   368.1    .045       0   383.1     .12       0
Bank Sta=368.1,383.1
XS Rating Curve= 0 ,0
Exp/Cntr=0.3,0.1

Type RM Length L Ch R = 1 ,42284.3 ,251.3,252.2,252.6
XS GIS Cut Line= 3
      2367317.27      382377.662      2367695.87      382220.848
     2368077.903      382072.615
#Sta/Elev= 30
       0  626.88    35.8  623.22    55.7  619.76    83.6  611.28   123.3  596.92
   171.1  584.23   214.8  568.75   234.7   567.5   310.3  566.06   346.1  562.94
   389.9  564.47   406.8     562   413.8  561.17   425.7  562.17   441.6  566.53
   453.6   574.1   473.4  588.73   485.4  596.16   501.3  604.29   541.1  622.45
   588.8  639.48   616.7  651.98   668.4  672.65   680.3  678.28   704.2  684.56
  721.56692.3439   767.8  701.86  782.26 701.047   795.7  699.16   819.6  698.22
#Mann= 5 ,-1 , 0
       0     .12       0   406.8    .045       0   425.7     .12       0
  721.56     .08       0  782.26    .016       0
Bank Sta=406.8,425.7
XS Rating Curve= 0 ,0
Exp/Cntr=0.3,0.1

Type RM Length L Ch R = 1 ,42032.1 ,236.2,236.7,236.8
XS GIS Cut Line= 2
      2367403.76      382592.925     2368049.619      382355.385
#Sta/Elev= 30
       0  638.73    35.8   635.8    75.6  630.81   115.4  622.81   135.2  617.79
   151.2  612.51     171  604.48   206.8   586.8   238.7  573.28   246.6  567.56
   250.6  565.55   266.5  560.81   278.4  559.67   286.4  561.56   294.4  562.28
   342.1   561.8     350   560.5     362   562.3   397.8  562.61   417.7   560.2
   433.8  560.34   441.5  561.63   461.4  578.84   497.2  598.12   521.1  609.69
   548.9  621.07   568.8  628.07   624.5  652.22   668.3  666.88   688.2  671.71
#Mann= 3 ,-1 , 0
       0     .12       0   417.7    .045       0   433.8     .12       0
Bank Sta=417.7,433.8
XS Rating Curve= 0 ,0
Exp/Cntr=0.3,0.1

Type RM Length L Ch R = 1 ,41795.4 ,171,175.2,178.8
XS GIS Cut Line= 3
     2367552.657      382683.076     2367662.249      382730.819
     2368142.935      382570.229
#Sta/Elev= 30
       0  621.36    27.9  616.31    47.8  610.86    87.7  595.01   119.5  580.56
   131.5   578.3   143.5  573.16   175.4  562.01   199.4  558.11   211.3  560.81
   219.3  560.29   231.3  557.77   239.3  559.36   255.2  560.16   267.2  559.43
  272.93  558.29   287.1  557.76   295.1  558.61   311.1  560.01   319.1  559.38
     331   560.7     347  560.65     359  561.67     367  563.75   394.9  577.72
   418.8  587.42   442.8  595.65   550.5  641.22   586.4  653.22   626.3  662.56
#Mann= 3 ,-1 , 0
       0     .12       0  272.93    .045       0   295.1     .12       0
Bank Sta=272.93,295.1
XS Rating Curve= 0 ,0
Exp/Cntr=0.3,0.1

Type RM Length L Ch R = 1 ,41620.2 ,179.3,172.7,165.8
XS GIS Cut Line= 4
     2367703.482      382909.856     2367795.712      382849.092
     2367947.622       382820.88     2368114.723       382741.67
#Sta/Elev= 30
       0  588.95    39.4  573.25    51.3  567.51    63.1  561.19    67.1  560.15
      75  559.53    90.7  559.75    98.6  561.18   110.4  564.62   114.4  565.01
   118.4  563.98   126.3  558.88   130.3  557.95   150.1  557.33     162  556.28
   169.9   555.1   177.8  554.66   188.1  555.23   205.5  557.32   217.4  557.79
   233.3  559.43     257   559.7   276.8  561.57   284.6  563.11   304.3  570.24
   347.6  591.42   371.2  601.84   398.7  613.04   426.3  623.27   449.9  632.61
#Mann= 3 ,-1 , 0
       0     .12       0   169.9    .045       0   188.1     .12       0
Bank Sta=169.9,188.1
XS Rating Curve= 0 ,0
Exp/Cntr=0.3,0.1

Type RM Length L Ch R = 1 ,41447.5 ,363.3,360.3,357.4
XS GIS Cut Line= 2
     2367562.541      383176.421       2368299.9      382799.866
#Sta/Elev= 30
       0  627.63      24  627.13      96  620.56     124  619.07     152  619.48
     168     618     192  608.74     220  595.15     264  570.05     280  558.48
     284  556.46     364  555.58     380  556.27     388  555.69   395.5  553.54
     404  553.04     416  553.63     424  555.25     440  555.07     452  557.86
     500  558.59     516  560.23     536  567.74     568  584.53     616  607.23
     660  621.61     716  643.75     756  655.95     776  663.29   827.9  669.71
#Mann= 3 ,-1 , 0
       0     .12       0   395.5    .045       0     416     .12       0
#XS Ineff= 2 , 0
                          451.86          559.64
Permanent Ineff=
       F       F
Bank Sta=395.5,416
XS Rating Curve= 0 ,0
Exp/Cntr=0.3,0.1

Type RM Length L Ch R = 1 ,41087.2 ,392,392.9,393.9
XS GIS Cut Line= 2
      2367704.23      383514.741     2368413.325      383069.438
#Sta/Elev= 30
       0  650.15    63.8  647.31   111.6  641.55   135.6  637.88   203.4  623.88
   227.3  616.85   263.2  603.73     311  584.27   358.8  562.24   374.8  556.97
   390.8  553.88   398.7  550.12   402.7  549.18   418.4   549.8   426.6  552.66
   430.6  553.06   454.6  551.94   466.5  553.04   478.5  552.36   530.3  558.17
   550.2  566.12   586.1  587.56     610   600.5     638  613.16   669.9  622.92
   709.7  638.89   765.6  658.65   781.5  662.05   813.4  670.88   837.3  674.62
#Mann= 3 ,-1 , 0
       0     .12       0   398.7    .045       0   418.4     .12       0
Bank Sta=398.7,418.4
XS Rating Curve= 0 ,0
Exp/Cntr=0.3,0.1

Type RM Length L Ch R = 1 ,40694.3 ,175,176,175.8
XS GIS Cut Line= 2
     2367905.749      383777.437     2368548.751      383426.349
#Sta/Elev= 30
       0   652.9    27.9   648.3    35.8  646.18   127.4  614.74   155.3  604.06
   171.2  596.46   199.1  584.62   242.9  568.84   282.7  551.97   298.6  549.89
   342.4  550.25   374.3  548.77   398.2  549.37     426  547.97     434  546.59
   445.9   544.9   453.9  545.75   457.9  549.37   465.8  560.87   469.8  565.18
   481.8  574.87   493.7   582.2   537.5  603.79   561.4  613.56   577.3  617.87
   593.2  623.32     641  644.49   668.9  655.02   692.8  662.25   732.6  671.76
#Mann= 3 ,-1 , 0
       0     .12       0     434    .045       0   453.9     .12       0
#XS Ineff= 2 , 0
          330.68  554.64
Permanent Ineff=
       F       F
Bank Sta=434,453.9
XS Rating Curve= 0 ,0
Exp/Cntr=0.3,0.1

Type RM Length L Ch R = 1 ,40518.4 ,356.5,357,357.6
XS GIS Cut Line= 3
      2367983.43      383838.675     2368167.615      383824.959
     2368700.575      383532.692
#Sta/Elev= 30
       0  641.08   176.8  593.45   216.7  579.65   232.7  572.82   248.7   568.3
   268.7  558.15   272.7  556.91   300.7  552.04   320.7   550.9   340.6  547.36
   352.6  548.55   376.1  543.49   388.6  543.07   392.6  543.36   416.6  548.48
   420.6   550.5   432.6  559.74   460.6  578.54   496.6  600.91   516.6   610.9
   572.6  634.08   612.6  648.82   644.6  658.72   660.6  663.04   676.6  665.68
  710.48 673.339   720.6  674.52   740.6  673.83  748.77674.4833   792.5  672.17
#Mann= 5 ,-1 , 0
       0     .12       0   376.1    .045       0   392.6     .12       0
  710.48    .016       0  748.77     .12       0
Bank Sta=376.1,392.6
XS Rating Curve= 0 ,0
Exp/Cntr=0.3,0.1

Type RM Length L Ch R = 1 ,40161.4 ,227.7,226.3,224.8
XS GIS Cut Line= 3
     2368150.841      384228.059     2368589.983       384000.35
      2368885.59      383861.331
#Sta/Elev= 30
       0  621.03    43.9  612.49    59.8  612.75   111.7  607.73   131.6  603.88
   147.6  605.14   199.5  599.14   239.4  577.51   283.2  551.29   299.2   545.8
   319.1   543.3     387  542.68   404.6  539.06   418.9  538.04   426.8  539.82
   434.8  545.58   458.8  568.84   474.7  579.11   498.6  593.05   530.5  606.13
   554.4  618.97   586.3  632.61   602.2  637.66   693.8  661.14  704.62663.0159
  739.17662.5956   753.6  663.68   777.5  661.03   789.5   661.6   821.3  658.98
#Mann= 5 ,-1 , 0
       0     .12       0   404.6    .045       0   426.8     .12       0
  704.62    .016       0  739.17     .12       0
#XS Ineff= 2 , 0
          363.29  546.12
Permanent Ineff=
       F       F
Bank Sta=404.6,426.8
XS Rating Curve= 0 ,0
Exp/Cntr=0.3,0.1

Type RM Length L Ch R = 1 ,39935   ,327.3,345.7,364.1
XS GIS Cut Line= 3
     2368200.797      384352.318     2368482.561      384320.446
     2368899.228       384068.71
#Sta/Elev= 30
       0  633.54      16     634      32  628.09    43.9  627.08    55.9  624.42
   115.8  616.53   199.7  603.29   219.7  597.09   247.6  585.34   283.6  567.69
   319.5   548.1   331.4   543.9   339.4  541.89   355.4  540.39   407.3  538.54
   419.8  536.44   431.2  536.33   443.2  536.77   451.2  540.24   467.1   553.4
     495  569.69     523  584.14   578.8  609.69   630.7  627.45   650.7   631.8
   702.5  646.34  716.56649.2402   734.5  652.62  755.51652.3145   770.4  652.51
#Mann= 5 ,-1 , 0
       0     .12       0   419.8    .045       0   443.2     .12       0
  716.56    .016       0  755.51     .12       0
Bank Sta=419.8,443.2
XS Rating Curve= 0 ,0
Exp/Cntr=0.3,0.1

Type RM Length L Ch R = 1 ,39589.3 ,214.4,221.1,227.6
XS GIS Cut Line= 3
     2368201.335      384431.571     2368737.553      384581.948
     2368859.081      384624.265
#Sta/Elev= 30
       0  632.65    11.9  629.51    27.8  628.04    63.6  622.61   103.4  613.98
   127.3  607.57   147.2  604.22   194.9  587.77   242.6  568.77   258.6   563.4
   270.5  556.57   294.4   545.8   314.2  540.96   346.1  536.22   385.9  537.77
   413.7  537.18   429.6  534.48   457.5     536   472.9  532.42   477.4   531.9
   487.9  532.63   493.3  534.28   517.1  556.64   525.1   562.8     537  570.98
   560.8  584.89   576.4  593.26     631  619.79   654.4  629.58   685.6  640.78
#Mann= 3 ,-1 , 0
       0     .12       0   472.9    .045       0   487.9     .12       0
Bank Sta=472.9,487.9
XS Rating Curve= 0 ,0
Exp/Cntr=0.3,0.1

Type RM Length L Ch R = 1 ,39368.2 ,412.8,399.7,386.5
XS GIS Cut Line= 2
     2368156.365      384503.982     2368874.828      384950.817
#Sta/Elev= 30
       0  636.53    55.9   621.3    91.8  607.13   179.6  569.95   211.5  558.94
   275.4  540.31   287.4  535.14   295.3  533.95   327.3  532.16   347.2  532.28
   359.2  533.57   403.1  533.65   427.3  530.81     435  530.68   442.3  530.95
     451  534.27   466.9  537.62   486.9   545.1   534.8  566.36   578.7  589.13
   586.7  592.44   622.6  602.32   662.5  611.62   682.4  617.75   710.4  622.68
   738.3  626.65   786.2   632.1   802.2  634.68   826.1  635.28   846.1  636.96
#Mann= 3 ,-1 , 0
       0     .12       0   427.3    .045       0   442.3     .12       0
Bank Sta=427.3,442.3
XS Rating Curve= 0 ,0
Exp/Cntr=0.3,0.1

Type RM Length L Ch R = 1 ,38968.5 ,267.9,259.8,251.6
XS GIS Cut Line= 3
     2368030.087      385040.932     2368598.642      385025.983
     2368834.124      384959.552
#Sta/Elev= 30
       0  662.04    75.6  623.71    95.4  612.89   123.3   596.7   139.2  586.21
   151.1  580.21   163.1  572.72   186.9   559.4   210.8   547.6   222.7  539.79
   234.7   537.6   254.6  527.55   266.5  526.35   278.4  527.99   290.3  529.53
     346  529.24   417.6  530.64   429.6  529.84   457.4  531.59   485.2  531.71
   493.2   532.8   513.1  539.87   544.9  553.17   580.6  565.71   608.2  574.43
   663.5  588.54   750.3  613.14   762.1  614.22     774  619.15   813.4  629.11
#Mann= 3 ,-1 , 0
       0     .12       0   254.6    .045       0   278.4     .12       0
#XS Ineff= 2 , 0
                          414.63          536.33
Permanent Ineff=
       F       F
Bank Sta=254.6,278.4
XS Rating Curve= 0 ,0
Exp/Cntr=0.3,0.1

Type RM Length L Ch R = 1 ,38708.7 ,390.7,378.4,363
XS GIS Cut Line= 2
     2368044.672      385398.228     2368844.975      385070.229
#Sta/Elev= 30
       0   660.1   20.74659.6675    47.8  656.52    59.8  653.72    71.7   649.2
    95.7  636.98   203.3   574.1   223.2  564.47   243.1  556.66   354.7  525.16
   366.7  526.73   394.6  527.05   418.5  526.69   430.5  524.65   442.4  524.06
   451.4  524.71   462.4  526.04   474.3  525.26   490.2   530.5   506.2  530.61
   534.1  532.72     554   535.7   581.9  544.68   617.8  559.16   633.7  563.39
   661.6  575.37   713.4  593.34   745.3  601.37   809.1  614.77   864.9  624.58
#Mann= 4 ,-1 , 0
       0    .016       0   20.74     .12       0   430.5    .045       0
   451.4     .12       0
Bank Sta=430.5,451.4
XS Rating Curve= 0 ,0
Exp/Cntr=0.3,0.1

Type RM Length L Ch R = 1 ,38330.3 ,298,289.3,280.5
XS GIS Cut Line= 2
     2368298.486      385802.629     2368902.648      385146.517
#Sta/Elev= 30
       0  654.32   10.81652.6953      68  643.09      96  633.52     116  628.76
     148  618.94     172  609.23     220  583.98     260  567.38     332  539.43
     360  526.59   386.4   520.2     396  519.92   401.4  520.17     416  523.96
     444  523.13     460  524.56     496  523.04   519.9  525.65   571.9  527.81
   583.9  529.65   603.9  535.96   687.9  573.28   727.9  589.08   811.9  611.46
   823.9   616.4  833.29618.7997   863.9  619.99  875.43625.6985   891.9  629.19
#Mann= 6 ,-1 , 0
       0     .06       0   10.81     .12       0   386.4    .045       0
   401.4     .12       0  833.29    .016       0  875.43     .12       0
Bank Sta=386.4,401.4
XS Rating Curve= 0 ,0
Exp/Cntr=0.3,0.1
